--- HECRAS_v1.prj (project) ---

Proj Title=HECRAS_v1
Current Geom=g01
Default Exp/Contr=0.3,0.1
SI Units
Geom File=g01
Y Axis Title=Elevation
X Axis Title(PF)=Main Channel Distance
X Axis Title(XS)=Station
BEGIN DESCRIPTION:
END DESCRIPTION:
DSS Export Rating Curves= 0
DSS Export Rating Curve Sorted= 0
DSS Export Volume Flow Curves= 0
DXF OffsetX= 0
DXF OffsetY= 0
DXF ScaleX= 1
DXF ScaleY= 10

--- HECRAS_v1.g01 (geometry) ---

Geom Title=HECRAS_v1
Program Version=5.01

Junct Name=1
Junct Desc=, 0 , 0 ,-1 ,0
Up River,Reach=ARROYOELZORRO   ,ARRIBALAT1
Dn River,Reach=ARROYOELZORRO   ,ABAJOLAT1
Junc L&A=0,0

River Reach=ARROYOELZORRO   ,ARRIBALAT1
Reach XY= 30
    1080707.4374    1573339.5833    1080687.7523    1573349.7434
    1080636.3172     1573396.416    1080550.5921    1573432.2935
    1080519.1595     1573427.531    1080513.4445     1573418.641
    1080528.0495    1573365.6184    1080525.5095    1573345.6159
     1080519.477    1573340.2184    1080492.1719    1573342.1234
    1080422.9568    1573444.6761     1080410.836    1573501.8389
    1080390.1985    1573530.9431    1080370.0901    1573533.8535
    1080237.7982    1573498.1347    1080173.2397    1573449.1867
     1080139.536     1573378.935    1080113.4599    1573351.9355
    1080078.0847    1573339.3843    1079986.1122    1573341.3699
    1079950.6469    1573323.7062    1079927.6034    1573291.4759
    1079900.9914    1573205.3105    1079862.9313    1573168.1895
     1079817.723    1573160.9037    1079670.7934    1573191.5554
     1079620.597    1573176.3569    1079592.4691    1573141.0177
    1079561.4908    1573047.1475    1079528.5191    1573013.8644

Type RM Length L Ch R = 1 ,10516.63,326.71,338.48,272.19
XS GIS Cut Line= 4
    1080327.0311    1572922.9204    1080508.3292    1573234.2431
    1080782.3396     1573544.788    1080904.0514    1573717.6348
#Sta/Elev= 30
       0   74.29   54.96      74  106.41   73.88  160.09    73.5  202.95      73
  239.59      73  296.77   72.81  373.39    72.5  413.09   72.16  508.37      72
  536.55    72.5  545.68    72.5   550.5      72  557.78      71  572.44      71
  580.98    71.5  596.55   72.06  605.68    72.5  618.98      74  631.62      75
  650.95    75.5  678.17    75.5  697.65   75.86  726.96    76.7  738.77   76.91
  773.94   77.38  802.87   77.49  859.15   78.02   891.6   78.11  985.81   77.95
#Mann= 0 , 0 , 0
Bank Sta=536.55,596.55
XS Rating Curve= 0 ,0
Exp/Cntr=0.3,0.1

Type RM Length L Ch R = 1 ,10178.15,130.71,126.74,122.71
XS GIS Cut Line= 4
    1080274.1143    1572941.9705    1080377.2263    1573318.1105
    1080566.5631    1573560.6676    1080749.9587    1573803.7037
#Sta/Elev= 30
       0   74.33   39.05      74  180.78    73.5  228.31      73  289.46      73
  440.96   72.08  469.28   72.24  474.55   72.38  482.82      72  493.37      71
  500.83    70.5  505.67    70.5  517.56    71.5  524.04    71.8  533.39      72
  651.94      72  667.53    71.5  707.05    71.5  732.02      72  737.33    72.5
  743.35    73.5  757.79   76.64  764.21    77.5  769.34   77.68  785.48   77.79
  815.14   77.43  832.97   78.09  850.74   78.47  939.19    79.5 1002.19      80
#Mann= 0 , 0 , 0
Bank Sta=469.28,533.39
XS Rating Curve= 0 ,0
Exp/Cntr=0.3,0.1

Type RM Length L Ch R = 1 ,10051.41,150.51,180.98,211.46
XS GIS Cut Line= 4
    1080240.2476    1572950.4372    1080352.9475    1573475.0008
     1080541.224    1573663.8071    1080671.8044    1573849.7252
#Sta/Elev= 30
       0      74   45.82      74  156.83    73.5  273.69   73.39  301.48      73
  319.19      73  358.67   72.56  373.11   72.66  378.61    72.5  572.77    72.5
  576.26    72.5  584.43      72  596.67   70.73  604.06   70.81  617.13    71.5
  632.85    71.5  659.99   71.73  697.24   71.51  724.75    71.1  739.02   71.24
  748.62    71.5  755.78      72  770.45      74  779.39   75.05  790.06   76.16
  798.65   76.84  812.08   77.59  839.05    78.5  912.04   79.54 1030.36   80.22
#Mann= 0 , 0 , 0
Bank Sta=572.77,632.85
XS Rating Curve= 0 ,0
Exp/Cntr=0.3,0.1

Type RM Length L Ch R = 1 ,9870.433,205.56,209.92,222.26
XS GIS Cut Line= 4
    1080202.1475    1572954.6705    1080254.1813     1573378.091
    1080194.4311    1573650.0588     1080377.746    1573958.0837
#Sta/Elev= 30
       0   73.68  266.43    73.5  301.61      73  353.82      73  454.44      72
  512.51      72  518.34      72  536.65      71  559.54      71  575.74   71.74
  586.02      72  594.87   71.31  604.48   71.04  621.28    71.5  637.17   71.53
   683.5    71.5  698.79      71  712.74      71  728.62    71.5  741.99   71.03
  753.58      71  823.39   71.69  889.07    71.5  910.13      72   934.4      72
  953.99   72.36 1022.46   72.58 1035.75      73 1045.59      74 1063.51   76.25
#Mann= 0 , 0 , 0
Bank Sta=512.51,575.74
XS Rating Curve= 0 ,0
Exp/Cntr=0.3,0.1

Type RM Length L Ch R = 1 ,9660.509,133.24,126.88,116.59
XS GIS Cut Line= 5
    1080161.9306    1572958.9446    1080152.5873    1573251.4818
    1080095.9811    1573338.1023    1079991.8435    1573479.1967
    1080234.5059    1573980.1218
#Sta/Elev= 30
       0   73.96   47.29    73.5  256.84    73.5  273.09      73  359.35   72.27
  376.51   72.03  389.93    70.5  415.39   70.84   423.7   70.49  427.79   71.21
  430.69   70.71  448.34   71.97  502.86   71.98  524.29   73.47  600.56      75
  746.21   76.39  787.41      76  821.77   74.34  862.37   75.47  922.19   76.04
  974.68    77.1  989.65    76.5 1001.61      75 1013.29      75 1046.13   77.49
 1061.74      78 1075.93    77.5 1099.93    75.7 1117.14      77 1128.13   78.98
#Mann= 0 , 0 , 0
Levee=0,,,-1,524.29,73.47035,,	339
Bank Sta=359.35,448.34
XS Rating Curve= 0 ,0
Exp/Cntr=0.3,0.1

Type RM Length L Ch R = 1 ,9533.624,62.94,98.04,133.14
XS GIS Cut Line= 5
    1080109.3166     1572950.726    1080050.9978    1573155.8972
     1079943.577     1573386.726    1079923.5675    1573427.4895
    1079827.7994    1574025.7831
#Sta/Elev= 30
       0    73.5   78.34   73.28   106.5      73  187.46   72.73  207.56   72.75
  209.43   73.36  233.88   73.36  254.88   71.86  369.71   71.86  390.29   70.38
  430.04   70.38  451.65   71.86  464.08   71.86  485.08   73.36  509.48   73.36
  512.06    72.5  536.06    72.5  590.18   73.69  601.72   73.86  628.31   73.91
   666.3   73.77  711.47   73.95  741.98   74.19  789.41      75  851.53   76.74
  915.75   78.01  970.82   78.53 1054.62   79.15 1088.83   79.48 1119.22   79.91
#Mann= 0 , 0 , 0
Levee=-1,233.88,73.36314,-1,485.08,73.36273,	340,	339
Bank Sta=369.71,451.65
XS Rating Curve= 0 ,0
Exp/Cntr=0.3,0.1

Type RM Length L Ch R = 1 ,9435.588,137.8,102.69,67.58
XS GIS Cut Line= 4
    1080083.4932    1572937.8142    1079991.2064    1573234.1482
     1079861.851     1573271.218    1079719.4258    1574024.0897
#Sta/Elev= 30
       0    73.3  207.07    72.5  209.48   73.32   234.1   73.33  255.29   71.83
   346.7   71.79   367.7   70.29   407.7   70.29   428.7   71.73  513.46   71.74
  535.12   73.25   560.3   73.25  565.65   71.66  578.22   71.33   591.3    70.5
   617.6   70.37  637.36   71.04  670.92   71.36  690.23   71.23  705.96   70.65
  721.87   70.44  730.54   70.74  745.07      72   766.4      72  780.24    71.5
  807.22    71.2  865.68   72.86  971.08      77 1040.58   77.99 1211.16   79.74
#Mann= 0 , 0 , 0
Levee=-1,234.1,73.32671,-1,535.13,73.24612,	340,	339
Bank Sta=346.7,428.7
XS Rating Curve= 0 ,0
Exp/Cntr=0.3,0.1

Type RM Length L Ch R = 1 ,9332.896,141.46,114.69,87.92
XS GIS Cut Line= 3
    1079992.4764    1572899.5025    1079778.3077     1573359.714
    1079621.0007    1574009.6964
#Sta/Elev= 30
       0      73  201.91    72.5  203.94   73.18  228.34   73.18  249.34   71.68
  257.43   71.68  278.72   70.19  318.56   70.19  339.62   71.68  458.54   71.68
  479.54   73.18  503.94   73.18  505.77   72.57  648.86    72.5  666.35   71.91
  673.85    71.5  717.72    70.5  725.81      70  758.58      70   785.2   70.77
  800.92   71.65  821.67   71.28  838.01      72  853.74    72.5  875.49    73.5
  910.34    75.5  941.61    76.5 1025.97   77.52 1084.68   78.49 1176.35   79.44
#Mann= 0 , 0 , 0
Levee=-1,228.34,73.17561,-1,479.54,73.17561,	340,	339
Bank Sta=257.43,339.62
XS Rating Curve= 0 ,0
Exp/Cntr=0.3,0.1

Type RM Length L Ch R = 1 ,9218.207,100.72,127.49,154.26
XS GIS Cut Line= 5
    1079875.0012    1572860.7674    1079739.5342    1573104.6079
    1079763.8079    1573214.4359    1079771.7076    1573257.0082
    1079542.2605    1573998.6897
#Sta/Elev= 30
       0   73.08  188.03   72.78  189.26   72.78  189.98   73.02  214.44   73.01
   235.5   71.51  309.42   71.53  330.42   70.08  370.42   70.08  391.42   71.58
  476.37   71.62  497.57   73.13  522.19   73.13  524.11    72.5  655.81   72.21
  674.96      72  787.28      72  797.42   70.99  815.41    69.5   822.6    69.5
  830.87      70  839.26      71  849.81   71.97  872.36   71.31  889.48    71.4
  925.24   72.48  954.33   73.74 1077.82    77.5 1132.44    78.5 1211.08   79.32
#Mann= 0 , 0 , 0
Levee=-1,214.44,73.01493,-1,497.56,73.12814,	340,	339
Bank Sta=309.42,391.42
XS Rating Curve= 0 ,0
Exp/Cntr=0.3,0.1

Type RM Length L Ch R = 1 ,9090.717,68.21,102.45,136.69
XS GIS Cut Line= 3
    1079795.4143     1572828.594    1079590.7473    1573268.3881
    1079386.4735    1573974.1363
#Sta/Elev= 30
       0   73.38  116.52      73  206.87      73  208.66   72.99  230.48   71.43
  349.22   71.43  370.18   69.96  410.01   69.97  431.31   71.43  439.68   71.43
  460.68   72.93  485.08   72.93   485.9   72.67  548.67   72.35  701.25   71.86
  714.03    71.5  732.03      70  742.52    69.5  759.73    69.5  764.57      70
  775.42    71.5  783.49   72.07  859.84      72  901.93   73.55  922.59   75.16
  930.92   75.68   951.4    76.5  964.59   76.83 1012.64   77.51  1219.8   79.36
#Mann= 0 , 0 , 0
Levee=-1,209.48,72.93304,-1,460.68,72.93301,	340,	339
Bank Sta=349.22,431.31
XS Rating Curve= 0 ,0
Exp/Cntr=0.3,0.1

Type RM Length L Ch R = 1 ,8988.263,137.11,103.08,68.73
XS GIS Cut Line= 4
    1079759.8543     1572810.814     1079645.554    1573077.6204
    1079521.3471    1573116.0751    1079286.2491    1573950.7471
#Sta/Elev= 30
       0   73.49  159.73   73.02  207.05   73.16  231.71    71.4  319.07   71.37
  340.07   69.87  380.07   69.87  401.07    71.3  484.52    71.3  508.09   72.96
  606.87   72.78   753.5      72  762.21    71.5  769.83      70  785.04   69.85
  811.06    70.5  823.24   72.36   839.2      73   852.1      73  864.25    72.5
   873.1    72.5  884.88    71.5  906.35      72  919.57   72.52     956   74.76
  977.07    75.8 1012.99      77  1035.4   77.48 1261.22      79 1287.43      79
#Mann= 0 , 0 , 0
Levee=-1,210.7,72.89437,-1,505.8,72.80102,	340,	339
Bank Sta=319.07,401.07
XS Rating Curve= 0 ,0
Exp/Cntr=0.3,0.1

River Reach=LATERAL1        ,LATERAL1
Reach XY= 30
    1081518.2289    1570397.8927    1081511.8789    1570446.5761
    1081461.9254    1570477.9029    1081153.9498    1570449.5395
    1081055.5246    1570500.3396    1081080.9247    1570687.0299
    1080962.8144    1570866.1003    1080974.8794    1570928.9654
    1081079.6547    1571054.6957    1081159.0298    1571260.4361
    1081169.1898    1571352.5113    1081112.6747    1571549.9967
    1081025.0445    1571595.7168    1080818.6691    1571610.3218
     1080738.024    1571650.3269    1080469.4184    1571690.9669
     1080494.501     1571945.285    1080595.1487    1572107.2103
    1080410.6808    1572306.9182    1080314.1606    1572330.7307
    1080193.5104    1572296.1232    1080067.1451    1572348.5108
    1079951.8924     1572216.748    1079907.7598     1572209.763
    1079755.9945    1572323.4282    1079699.7969    1572415.5034
    1079697.2569    1572607.9088    1079609.6267    1572706.0165
    1079550.5716    1572842.8593    1079526.3885    1573012.8008

Type RM Length L Ch R = 1 ,4571.366,152.41,163.43,174.48
XS GIS Cut Line= 4
    1081393.6367    1570101.9591     1081441.199    1570332.9487
    1081520.5742    1570623.9909    1081860.0449    1570801.3279
#Sta/Elev= 28
       0      79   22.59      79  119.12   79.41  216.56    79.5  273.55   79.16
  285.76      79  335.51   78.85  350.79   78.54  352.15    78.5  357.99      78
   368.3    76.5  374.48      76   391.7      76  396.05    76.5  402.91    77.5
   410.8    78.3  413.09    78.5  460.85    79.5   472.3      80  516.74      81
  536.76    81.1  568.37    81.5  668.54   82.38  703.02    82.5  749.23   82.82
  843.89   83.17   874.3    83.1  920.51   83.14
#Mann= 0 , 0 , 0
Bank Sta=350.79,410.8
XS Rating Curve= 0 ,0
Exp/Cntr=0.3,0.1

Type RM Length L Ch R = 1 ,4407.936,443.54,396.03,348.49
XS GIS Cut Line= 4
    1081253.6858     1570142.195    1081335.3655    1570306.4903
    1081306.8387     1570585.175    1081790.6318    1570939.9528
#Sta/Elev= 30
       0   78.85   44.52      79  246.94      79  257.12   78.65  265.78    78.6
  274.62   78.71  296.55   78.78  309.08    78.5  317.63   78.02  319.66   77.82
  322.92    77.5  329.69    76.5  336.34      76  360.94      76  367.68    76.5
  372.39   76.98  378.77      78  380.37   78.12  385.27    78.5  425.28    78.5
   478.3   79.51  508.98      80  529.77      80  559.12   80.24   611.4    80.5
  756.96      81  819.72   81.47  888.71   81.85 1028.57   82.11 1063.56   82.01
#Mann= 0 , 0 , 0
Bank Sta=319.66,380.37
XS Rating Curve= 0 ,0
Exp/Cntr=0.3,0.1

Type RM Length L Ch R = 1 ,4011.903,127.44,145.59,163.74
XS GIS Cut Line= 4
    1080708.7383    1570491.5304    1080921.5307    1570597.1121
    1081192.4902    1570621.3451    1081748.8517    1571024.5408
#Sta/Elev= 30
       0   77.12  187.64    77.9  314.07      78  348.21   78.19  353.85   78.07
  354.92      78  358.17    77.5  369.27   75.51   373.9      75     397      75
  412.29   76.51  418.41   76.94  425.44   77.13  431.74    77.5  452.77      78
  464.98   77.77  475.06   77.75  490.37   77.78  498.14      78  532.95      78
     576      79  631.16   79.56  695.41   79.84  837.48   80.21  872.46   80.47
  920.67    80.5  955.68   80.67 1106.34   80.85 1153.18   81.02 1196.69   80.89
#Mann= 0 , 0 , 0
Bank Sta=353.85,418.41
XS Rating Curve= 0 ,0
Exp/Cntr=0.3,0.1

Type RM Length L Ch R = 1 ,3866.315,225.37,200,174.75
XS GIS Cut Line= 4
    1080660.7755    1570590.9984    1080958.4221    1570667.3234
    1081175.4436    1570853.3408    1081659.8275    1571156.3035
#Sta/Elev= 30
       0   77.02  107.61    77.5  231.58    77.7  308.02   77.99  335.73      78
  361.51   77.52  374.15      77  395.57   76.54  398.75   76.37  403.98      76
  414.38      75  440.59      75  443.95    75.5  451.88   76.99  455.46    77.5
  458.75    77.5  491.12    77.5  523.92   77.65  547.09    77.5  577.54   77.62
  605.73      78   648.6   78.24  781.16   78.69  819.93   78.92  842.05   78.93
  884.91   79.19  1003.6   79.49 1049.65   79.35 1109.03   78.86 1164.44   78.91
#Mann= 0 , 0 , 0
Bank Sta=398.75,458.75
XS Rating Curve= 0 ,0
Exp/Cntr=0.3,0.1

Type RM Length L Ch R = 1 ,3666.315,208.53,200,191.35
XS GIS Cut Line= 4
    1080591.5109    1570888.9546    1080787.6296    1570935.8453
     1081141.525    1570888.6593    1081641.6243    1571220.7033
#Sta/Elev= 30
       0   76.87   25.29      77  214.53      77  278.02   77.15  314.66   77.31
  334.66    77.5  353.25    77.5  362.73      77  365.18    76.5  373.23    74.5
  390.54    74.5  404.18    75.5  414.05   76.47  421.85      77  491.43    77.5
  620.24    77.5  668.23   77.92  719.59      78  751.34    78.4  758.02   78.39
  771.36   78.18  788.64   78.16  808.24   78.28   823.6    78.5  872.58   78.62
  947.16   78.97  977.67   78.94 1010.47   78.79 1063.58   78.26 1158.97   78.17
#Mann= 0 , 0 , 0
Bank Sta=353.25,414.05
XS Rating Curve= 0 ,0
Exp/Cntr=0.3,0.1

Type RM Length L Ch R = 1 ,3466.315,196.37,200,203.63
XS GIS Cut Line= 4
     1080606.752    1571080.9971    1080921.7505    1571143.2625
    1081221.8512    1571010.8655    1081624.2068    1571282.5043
#Sta/Elev= 30
       0   75.86   114.1   76.03  214.64    76.5  319.04   76.74  366.74      77
  471.31      77  473.26      77  478.48    76.5   489.7    74.5  494.18      74
  509.17      74  514.75    74.5  522.46      76  525.79    76.5  531.31    76.8
  535.57      77  584.65      77  607.19    77.5  734.46    77.5  764.18   77.71
  801.81   77.78  826.41   78.04  897.13   78.31  957.89   78.16  994.72   77.81
  1012.4   77.74 1050.79   77.73 1083.48   77.51 1109.79   77.21 1134.57   77.17
#Mann= 0 , 0 , 0
Bank Sta=471.31,531.31
XS Rating Curve= 0 ,0
Exp/Cntr=0.3,0.1

Type RM Length L Ch R = 1 ,3266.315,184.79,200,215.21
XS GIS Cut Line= 4
    1080595.0101    1571256.4086    1080957.9986    1571317.8097
    1081316.1518    1571209.0849    1081593.8293    1571399.4434
#Sta/Elev= 30
       0    75.5   98.33    75.5  180.22      76  217.81   76.01  308.54    76.5
  344.18    76.5  429.31      77  495.72      77  506.44   76.49  511.56   76.37
  534.21   76.35  547.17   76.18  551.66      76  555.49   75.58  563.52    74.5
  568.16      74  574.91    73.5  583.66    73.5  589.15      74  600.69      76
  607.17   77.01  632.77   77.33  665.46      77  899.52   77.01   952.6   76.83
 1004.65   76.47 1026.74   76.01 1044.84      75 1065.64      76  1079.1   76.25
#Mann= 0 , 0 , 0
Bank Sta=547.17,607.17
XS Rating Curve= 0 ,0
Exp/Cntr=0.3,0.1

Type RM Length L Ch R = 1 ,3066.315,165.67,200,234.33
XS GIS Cut Line= 4
    1080510.4142    1571327.4268    1080932.1897    1571407.2786
    1081343.4433    1571495.4044    1081546.3129    1571648.9608
#Sta/Elev= 30
       0    75.5  141.84    75.5  249.87      76  301.21      76  374.81    76.5
     397    76.5  491.95      77  524.68      77   563.9   76.52  589.07    75.5
  622.19   75.07  632.03      75   648.1    73.5  654.41    73.5  661.02      74
  668.93      75   679.2    76.5  682.19   76.53  732.44   76.72  771.91    76.5
  811.96    76.5  850.64   76.31  888.68   76.01  932.18    75.5  947.53    74.5
  952.92    74.9  958.64    75.5 1029.37   75.76 1055.21      76 1104.29      76
#Mann= 0 , 0 , 0
Bank Sta=622.19,682.19
XS Rating Curve= 0 ,0
Exp/Cntr=0.3,0.1

Type RM Length L Ch R = 1 ,2866.315,192.19,200,207.81
XS GIS Cut Line= 4
    1080480.4185    1571356.0345    1080998.9119    1571452.4209
    1081074.7051    1571789.2748    1081372.5527    1572002.1389
#Sta/Elev= 30
       0    75.5  155.77    75.5  263.17      76  314.87      76  394.08    76.5
  508.65      77  540.95      77  596.73   76.51   628.7      76  636.94      76
  642.91   75.78  650.75    75.5  670.45    73.5  693.83    73.5  702.91   74.75
  711.22      76  721.63    76.5  737.08    76.5  798.23      76   880.5    75.5
  895.95   74.64   915.7   74.17   927.3    73.5  936.17    73.5  940.58      74
  947.45      75  952.29    75.5 1071.15    75.5 1101.27   75.63 1238.74   75.79
#Mann= 0 , 0 , 0
Bank Sta=642.91,702.91
XS Rating Curve= 0 ,0
Exp/Cntr=0.3,0.1

Type RM Length L Ch R = 1 ,2666.315,198.69,200,201.31
XS GIS Cut Line= 4
    1080413.8089    1571417.1216    1080837.3071    1571491.9031
     1080825.417    1571801.0496    1081227.9039    1572100.2957
#Sta/Elev= 30
       0    75.3   59.16    75.5   119.6    75.5  229.11      76  290.18      76
  416.36    76.5  490.59    76.5  509.01      76   519.1   75.45  530.54    74.5
  538.59   73.51  546.13      73  559.12      73  573.11   73.99   579.1    74.3
  591.04      75  600.21      76  609.19    76.5  623.05    76.5  680.09      76
  693.95      76  751.24   75.53  901.81   75.49  950.83      75  962.64    73.5
  968.92    73.5  981.86      75 1097.49   75.18 1187.19   75.13 1240.97   75.31
#Mann= 0 , 0 , 0
Bank Sta=519.1,579.1
XS Rating Curve= 0 ,0
Exp/Cntr=0.3,0.1

Type RM Length L Ch R = 1 ,2466.315,249.51,200,150.31
XS GIS Cut Line= 4
    1080356.2232    1571464.6942    1080655.8705    1571508.8005
    1080636.4999    1571737.3738    1081190.6132    1572157.6623
#Sta/Elev= 29
       0   75.05  129.25   75.53  231.45      76  414.03      76  417.14   75.93
  419.77   75.73  426.04      75  436.16    73.5  440.94      73  447.68    72.5
   458.7    72.5  466.35    73.5  468.97      74  475.54    75.5  478.49      76
  479.78   76.06  488.87   76.42   512.3   76.42  663.32   75.63  704.07    75.5
  783.39   75.34  887.13    75.3   925.6      75  931.26    74.5  935.05      74
   945.2      74  953.65      75 1153.43      75 1227.74    75.3
#Mann= 0 , 0 , 0
Bank Sta=419.77,479.78
XS Rating Curve= 0 ,0
Exp/Cntr=0.3,0.1

Type RM Length L Ch R = 1 ,2266.315,208.24,200,191.76
XS GIS Cut Line= 4
    1080212.2983    1571692.6391    1080255.2301    1571702.1731
    1080547.5626    1571712.6135     1081148.028    1572190.0326
#Sta/Elev= 30
       0   74.88  133.44   75.49  193.89      76  222.74      76  224.25   75.87
  228.63    75.5  235.47      74  238.21    73.5  242.68      73  248.74   72.62
  257.67   72.69     266      73  273.15    73.5  284.25   74.45  294.88    75.5
  308.28   75.97  341.67      76  375.91   76.24  473.47   76.08  559.14    75.5
  603.46    75.5  780.73      75  800.12    74.5  815.02    73.5  821.27    73.5
  834.08      75  926.78   74.91  932.61      75 1021.16      75 1103.63   75.29
#Mann= 0 , 0 , 0
Bank Sta=224.25,284.25
XS Rating Curve= 0 ,0
Exp/Cntr=0.3,0.1

Type RM Length L Ch R = 1 ,2066.315,211.93,200,188.07
XS GIS Cut Line= 4
    1080078.1307    1571881.4182    1080317.4153     1571947.621
    1080645.3778    1571866.6952    1081111.3766    1572231.5927
#Sta/Elev= 30
       0   74.52   211.7      75  300.93    75.5  391.45    75.5  395.62    75.5
  401.35      75   414.2      73  420.87    72.5  428.26    72.5  435.78      73
  444.61    74.5  451.45    75.2   455.9    75.5   509.2      76  564.57      76
  638.95    75.5  861.11      75  865.39    74.5  870.63    73.5  879.49   73.01
   883.8   73.32  891.84    74.5   897.7      75  951.24      75  966.65    74.5
  973.92    74.5 1003.67   74.96 1055.17      75 1127.66   75.46 1177.94    75.5
#Mann= 0 , 0 , 0
Bank Sta=391.45,451.45
XS Rating Curve= 0 ,0
Exp/Cntr=0.3,0.1

Type RM Length L Ch R = 1 ,1866.315,158.12,200,241.88
XS GIS Cut Line= 4
    1080035.6115    1571945.0255    1080541.2594    1572105.8958
    1080680.2679    1572002.6317    1081065.8008    1572304.3412
#Sta/Elev= 30
       0    74.5   72.07   74.54  205.82      75  217.69    75.5   230.6    75.5
  250.24      75  258.55      75  280.63    75.5  370.62    75.5  446.42      76
  476.36      76  555.16    75.5  559.14    75.5  564.22      75  574.28      73
  580.04    72.5  601.97    72.5  606.75      73  615.16   74.42  624.78   75.57
  720.93    75.5  790.11   75.07  839.99   74.57  871.58    74.5  875.56      74
  883.22    72.5  891.13    72.5  914.23    74.5 1082.12   74.84 1193.34   75.47
#Mann= 0 , 0 , 0
Bank Sta=555.16,615.16
XS Rating Curve= 0 ,0
Exp/Cntr=0.3,0.1

Type RM Length L Ch R = 1 ,1666.315,177.66,200,222.34
XS GIS Cut Line= 4
    1079970.6561    1571994.2082    1080329.7154    1572077.9904
    1080643.9976    1572369.1636    1080877.7629    1572548.1553
#Sta/Elev= 30
       0    74.5  227.76      75  309.06      75  317.96    75.2   368.7   75.47
  438.91    75.5  473.27      76  489.48      76  535.71    75.5  550.97    75.5
  556.53      75   567.8    72.5  572.23      72  577.77      72  590.06    72.5
   594.4      73  607.86      75  610.97   75.15  617.83    75.5  629.63    75.5
  734.54    74.5  801.84   74.19  940.24   73.87  991.57      74 1005.43   73.51
 1012.74    72.5 1022.07    72.5 1028.71    73.5  1033.1      74 1091.56      74
#Mann= 0 , 0 , 0
Bank Sta=550.97,610.97
XS Rating Curve= 0 ,0
Exp/Cntr=0.3,0.1

Type RM Length L Ch R = 1 ,1466.315,215.04,200,184.95
XS GIS Cut Line= 4
    1079900.4549     1572041.573    1080314.2202    1572157.3594
    1080340.1248     1572473.396    1080710.0367    1572753.1583
#Sta/Elev= 30
       0    74.5   62.68    74.5  145.72   74.84   234.9      75  349.11      75
  442.19   75.47   490.9    75.5  553.27    74.5  568.45   74.03  573.79   73.79
  580.24   73.51  586.69      73  593.86      72  610.69      72  616.73    72.5
  627.34      74  633.83   74.83  635.08      75  652.52      75  750.56    74.5
  770.29   74.48  883.71      74  915.67   73.98 1032.25    73.5 1159.98    73.5
  1169.9      72 1175.51   72.01 1184.89    72.5 1194.77    73.5 1210.55    73.5
#Mann= 0 , 0 , 0
Bank Sta=573.79,633.83
XS Rating Curve= 0 ,0
Exp/Cntr=0.3,0.1

Type RM Length L Ch R = 1 ,1266.315,410.51,400,389.53
XS GIS Cut Line= 4
    1079784.3397     1572071.356    1080040.1108    1572163.4889
    1080243.6466    1572472.3018    1080683.0551    1572807.7735
#Sta/Elev= 30
       0   74.33   55.54    74.5   208.2    74.5  258.86      75  311.83      75
  375.22    75.5  418.48   75.43   431.8   75.26  440.92      75  446.31      74
  453.08   72.48  455.92      72  460.55    71.5  467.82    71.5  474.04      72
  477.82    72.5  486.19      74  489.47    74.5   491.8   74.69  496.21      75
   619.2      75  719.12    74.5  973.75    73.5 1165.84    73.5 1173.76      73
 1178.08    72.5 1182.58   72.19 1187.11      72 1188.63    72.1 1194.54    72.8
#Mann= 0 , 0 , 0
Bank Sta=431.8,491.8
XS Rating Curve= 0 ,0
Exp/Cntr=0.3,0.1

Type RM Length L Ch R = 1 ,866.3152,209.16,200,190.8
XS GIS Cut Line= 3
    1079643.4541    1572112.7012    1080005.4348    1572386.9289
    1080630.2867    1572854.0753
#Sta/Elev= 30
       0      74   43.11      74   63.48   74.12  151.63      74  180.83    74.5
  219.59    74.5  222.51    74.5  227.04      74  237.66      72  241.66    71.5
  261.73    71.5  268.17    72.5  275.29      74  279.23    74.5     280    74.5
  350.02    74.5  376.43   74.64  423.64    74.5  434.65   74.65  486.71    74.5
  556.13    74.5  592.45   74.66  630.84      75  704.45      75  784.57    74.5
   859.9   74.27  997.48    73.5 1047.47    73.5 1194.83   73.13  1234.3   73.43
#Mann= 0 , 0 , 0
Bank Sta=219.59,280
XS Rating Curve= 0 ,0
Exp/Cntr=0.3,0.1

Type RM Length L Ch R = 1 ,666.3153,201.09,200,198.91
XS GIS Cut Line= 3
     1079545.912    1572344.5175     1079874.612    1572461.9099
    1080500.4923    1572908.3154
#Sta/Elev= 25
       0   73.68  138.79   74.49  141.01    74.5  148.02   74.02  151.99    73.5
  160.17    71.5  162.81      71  177.32      71  181.77   71.63  191.54    73.5
  195.51      74  198.79      74  273.97   74.16  307.56      74   437.4      74
  470.25   74.31  524.23    74.5   577.9    74.5  601.32   74.35   641.8    74.5
  840.62    74.5  848.79   74.71  862.69    74.5  935.95   74.49  1117.8   73.26
#Mann= 0 , 0 , 0
Bank Sta=138.79,198.79
XS Rating Curve= 0 ,0
Exp/Cntr=0.3,0.1

Type RM Length L Ch R = 1 ,466.3153,133.35,138.85,144.35
XS GIS Cut Line= 3
    1079485.0302    1572529.6118     1079885.609      1572655.92
    1080224.8188    1572885.3892
#Sta/Elev= 26
       0   73.45   48.82    73.5  147.69      74  188.66      74  195.95   73.58
  202.63      73  212.77    71.5  219.46      71  227.92      71  235.69    71.5
  244.38      73  248.04    73.5  253.15      74  255.95      74  316.28      74
  376.01    73.5  460.25    73.5     490   73.88  504.04   73.95  550.53    73.5
  599.18   73.42  633.96    73.5  736.37    73.5  792.01   74.18  816.14   74.27
  829.56   74.21
#Mann= 0 , 0 , 0
Bank Sta=195.95,255.95
XS Rating Curve= 0 ,0
Exp/Cntr=0.3,0.1

Type RM Length L Ch R = 1 ,327.4682,124.13,327.54,124.31
XS GIS Cut Line= 3
    1079445.6949    1572613.6877    1079779.4184    1572790.7109
    1080103.7223    1572902.2829
#Sta/Elev= 20
       0   73.19   43.77    73.5  158.42    73.5  167.88   73.47   172.2      73
  181.88      71  187.32    70.5  190.49    70.5  198.68      71   208.4      72
  218.41   73.44   219.8   73.58  224.86      74  243.24      74  357.09    73.5
     383    73.5  470.57   73.18  549.23      73  668.55   73.04  720.73   73.49
#Mann= 0 , 0 , 0
Bank Sta=158.42,219.8
XS Rating Curve= 0 ,0
Exp/Cntr=0.3,0.1

River Reach=ARROYOELZORRO   ,ABAJOLAT1
Reach XY= 30
    1079528.5191    1573013.8644    1079327.7203    1573037.6709
    1078910.1353    1572733.9715    1078253.1058    1572618.3051
    1078094.2524    1572733.3828     1077901.525    1572656.1992
    1077773.5463    1572795.8368    1077590.4555    1572744.3908
    1077195.6486    1573072.3463    1076992.2968    1573064.6889
    1076912.2578    1573236.1591    1076722.9953    1573202.6476
    1076612.4146    1573358.3916    1076411.5354    1573301.7432
     1076266.837    1573437.2883    1076101.9001    1573337.8544
    1075934.8719    1573443.2967    1075776.3981    1573325.9612
    1075314.2113    1573352.5123    1075021.8357    1573164.1616
    1074762.1036    1573307.0204    1074809.0672    1573474.3696
     1074606.396     1573339.961    1074509.6906    1573460.0821
    1074467.1477    1573329.4493    1074343.8516    1573398.9026
    1074180.2065    1573289.1003    1074303.8995    1573184.8543
    1074009.9468    1572948.0517    1073636.6961    1573264.4416

Type RM Length L Ch R = 1 ,8885.184,132.08,96,60.24
XS GIS Cut Line= 5
    1079689.4749    1572775.0158    1079573.3755    1572915.1394
    1079527.1627    1573013.1873     1079441.341    1573198.8588
    1079203.8048    1573913.9964
#Sta/Elev= 30
       0    73.7   68.38    73.5  207.42    73.5  240.31   71.24  249.34   71.24
  270.65   69.77  310.66   69.77  331.47   71.24  449.51   71.24  477.54   73.25
  510.44      73  597.78      73  699.99   72.01  722.46    70.5  739.33   70.27
  755.91    69.5  764.56    69.5  768.83      70  780.68      72  788.11    72.6
  802.42   72.93  815.94   72.83  827.78      73  856.22    71.5  863.31    71.5
  918.75    73.5  989.86    76.5 1026.76   77.38 1157.89    78.5 1248.47   78.74
#Mann= 0 , 0 , 0
Levee=-1,219.31,72.74111,-1,470.51,72.74126,	340,	339
Bank Sta=249.34,331.47
XS Rating Curve= 0 ,0
Exp/Cntr=0.3,0.1

Type RM Length L Ch R = 1 ,8789.181,71.26,107.16,143.04
XS GIS Cut Line= 5
    1079531.8761    1572688.6196    1079402.7592    1572950.0285
    1079453.2203    1573057.3448    1079460.9676    1573080.2037
    1079160.4004    1573894.0637
#Sta/Elev= 30
       0    73.5   212.4    73.5  246.26   71.08  328.15   71.11  349.15   69.68
  389.15   69.68  410.15   71.18  504.98   71.21  535.47   73.39  575.11      73
  669.62      73  708.06    72.5  721.73   71.19  730.62    70.5  744.79   70.14
  757.94    69.5  780.38    69.5  790.23   69.83  796.36   70.29  810.78   71.99
  817.23    72.5  879.82   72.37   890.5   72.16  906.69    71.5  927.06    71.5
  985.34   73.21 1044.39      76 1076.42   76.89 1227.07   78.49 1301.87    78.5
#Mann= 0 , 0 , 0
Levee=-1,225.26,72.58036,-1,526.05,72.71256,	340,	339
Bank Sta=328.15,410.15
XS Rating Curve= 0 ,0
Exp/Cntr=0.3,0.1

Type RM Length L Ch R = 1 ,8682.02 ,74.63,111.47,148.33
XS GIS Cut Line= 4
    1079486.3677    1572661.6321    1079419.3723    1572857.7406
    1079292.7963    1573129.7306    1079063.1393    1573850.2486
#Sta/Elev= 30
       0    73.5  218.95   73.47  252.64   71.05  367.49   71.05  388.54   69.58
  428.82   69.58  449.82   71.05  461.84   71.05  495.23   73.48  503.71    73.5
  511.46   73.01  525.43    70.5  534.64    69.5  571.54    69.5  577.94      70
  594.06    72.5   605.9   73.31  636.65      73  759.24      73  764.93    72.5
  775.55    70.5  782.78    69.5  796.46    69.5  827.74      72  869.52   71.79
  888.29      71  901.54      71 1081.42    76.5 1202.71   77.99 1263.47   78.16
#Mann= 0 , 0 , 0
Levee=-1,231.64,72.55075,-1,482.84,72.55075,	340,	339
Bank Sta=367.49,449.82
XS Rating Curve= 0 ,0
Exp/Cntr=0.3,0.1

Type RM Length L Ch R = 1 ,8570.554,128.33,91.45,54.52
XS GIS Cut Line= 6
    1079448.3734    1572649.6729    1079387.8709    1572843.0808
    1079344.2332    1572935.8468    1079236.2393    1572961.8225
     1079212.153    1572968.0202    1078982.7058    1573824.8486
#Sta/Elev= 30
       0   73.22   33.56   73.11  216.39   73.27  248.05   71.01  334.24   70.98
  355.24   69.48  395.24   69.48  416.24   70.91  509.33    70.9  537.96   72.92
  548.72      73  642.69   72.98  768.63    72.5  924.21    72.5  942.88      71
  954.78    69.5  963.72    69.5   971.2   69.18  980.22    69.5  986.24   70.17
  995.65    71.5 1003.15      72 1024.17   72.34 1039.11   72.73 1068.18    73.9
 1090.81    74.5 1137.54      76 1183.97      77 1307.88   77.99 1328.13   78.03
#Mann= 0 , 0 , 0
Levee=-1,227.05,72.51025,-1,530.65,72.40443,	340,	339
Bank Sta=334.24,416.24
XS Rating Curve= 0 ,0
Exp/Cntr=0.3,0.1

Type RM Length L Ch R = 1 ,8479.103,143.28,107.05,70.86
XS GIS Cut Line= 4
    1079359.4733    1572590.4061    1079272.7216    1572789.4938
    1079146.1456    1573061.4837    1078894.6523    1573793.5218
#Sta/Elev= 30
       0      73  124.03      73  236.91    72.7  262.57   70.86  270.55   70.86
  291.77   69.39  331.85    69.4  353.22   70.86  471.77   70.86  496.41   72.62
  515.77   72.68  600.11   72.76  786.04   72.12  939.38    72.5  958.72      72
  977.18    70.5  995.44    70.5 1008.04      70 1014.04    69.5  1024.6      69
 1036.88      69 1041.74   69.49 1056.77   71.46 1070.55    73.5 1078.59      74
 1092.19    74.5  1145.6      76 1225.17    77.5 1269.16      78  1291.2      78
#Mann= 0 , 0 , 0
Levee=-1,241.57,72.36261,-1,492.77,72.36261,	340,	339
Bank Sta=270.55,353.22
XS Rating Curve= 0 ,0
Exp/Cntr=0.3,0.1

Type RM Length L Ch R = 1 ,8372.053,72.42,108.66,144.91
XS GIS Cut Line= 6
    1079236.8122    1572529.6153    1079140.6199    1572728.0176
    1079096.0536    1572807.9575    1079149.5197     1572919.071
     1079160.612    1572940.2495    1078827.2364    1573784.8012
#Sta/Elev= 30
       0      73   60.21      73  129.66   72.54  240.63    72.5  266.01   70.69
  353.32   70.72  374.32   69.29  414.32   69.29  435.32   70.79  529.97   70.82
  553.46    72.5   631.7   72.63  725.27    72.5  844.52      72  984.74      72
 1014.89    72.4 1035.04   72.15 1067.22   71.13 1079.68    70.5 1107.13      70
 1116.99      69 1134.46      69  1138.6    69.5 1140.94      70  1151.6   73.25
 1159.01      74 1253.53   76.49 1306.77      77 1352.15      78  1367.2      78
#Mann= 0 , 0 , 0
Levee=-1,244.96,72.19109,-1,551.01,72.32472,	340,	339
Bank Sta=353.32,435.32
XS Rating Curve= 0 ,0
Exp/Cntr=0.3,0.1

Type RM Length L Ch R = 1 ,8263.394,75.89,111.57,147.24
XS GIS Cut Line= 4
    1079207.1788    1572509.5069    1079114.7195    1572715.9643
    1078988.1435    1572987.9543    1078734.1028    1573749.8761
#Sta/Elev= 30
       0      73   62.84    72.5  245.85    72.5  271.62   70.66  388.31   70.66
  409.19   69.19  449.23   69.19  470.35   70.66  480.82   70.66  501.82   72.16
  526.22   72.16  526.96   71.92  687.74      72  756.24   71.72 1014.35      72
 1024.78      71 1037.96      69 1045.76    68.5 1051.26    68.5 1060.57      69
 1094.21      72 1105.86      72 1118.71      71  1133.7   70.96 1159.07   71.82
  1185.9    73.5  1222.2      75 1243.25   75.26  1278.4   76.23 1329.37   76.96
#Mann= 0 , 0 , 0
Levee=-1,250.61,72.15994,-1,501.81,72.15994,	340,	339
Bank Sta=388.31,470.35
XS Rating Curve= 0 ,0
Exp/Cntr=0.3,0.1

Type RM Length L Ch R = 1 ,8151.827,132.49,93.75,55.01
XS GIS Cut Line= 6
    1079179.6621    1572494.6902    1079087.3428     1572703.224
    1079045.2535    1572789.9658    1078932.8887    1572820.4592
    1078914.0199    1572841.8243    1078634.6193     1573714.951
#Sta/Elev= 30
       0   72.91   47.57    72.5  247.93   72.45  273.46   70.62   358.9   70.59
   379.9   69.09   419.9   69.09   440.9   70.52  528.14   70.51   549.2   72.01
  573.68   72.02  575.23    71.5  694.23   71.71  827.29   71.31  1021.3   71.69
 1058.96   71.22 1110.43   71.93 1154.79      72 1178.52    71.5 1206.48   70.13
 1231.08   70.64 1280.53    68.5 1295.36    68.5 1308.85      69 1325.22    68.5
 1333.96      69 1342.84      70 1364.31   73.54 1374.45   74.56 1386.14      75
#Mann= 0 , 0 , 0
Levee=-1,252.46,70.9492,-1,549.29,72.01389,	340,	339
Bank Sta=358.9,440.9
XS Rating Curve= 0 ,0
Exp/Cntr=0.3,0.1

Type RM Length L Ch R = 1 ,8058.077,133.73,95.13,56.53
XS GIS Cut Line= 4
    1079064.8327    1572431.4018    1078954.4105    1572645.2909
    1078864.4802    1572883.4531     1078573.765     1573693.996
#Sta/Elev= 30
       0      73   28.62      73  102.26    72.5  122.09    72.5  150.84      72
  240.71   71.86  266.96   71.97  287.96   70.47  298.06   70.47  319.05      69
  359.06      69  380.13   70.47  497.16   70.47  518.16   71.97  542.56   71.97
  543.98    71.5  717.22    71.5  787.06   71.12  910.99    71.5 1080.33    71.5
 1192.41    71.9 1247.99   71.81 1272.48    71.5 1280.85    70.5 1293.84    69.5
 1316.32   68.71 1324.62   68.83 1335.22   69.37  1348.5      71 1356.39   71.61
#Mann= 0 , 0 , 0
Levee=-1,267.02,71.96507,-1,518.24,71.9697,	340,	339
Bank Sta=298.06,380.13
XS Rating Curve= 0 ,0
Exp/Cntr=0.3,0.1

Type RM Length L Ch R = 1 ,7962.949,78.48,114.34,150.19
XS GIS Cut Line= 6
    1078881.4231    1572348.1108    1078808.8085    1572598.7291
    1078784.9029    1572683.3915    1078852.9902    1572787.2213
    1078860.2564    1572814.6251    1078534.2891    1573687.5401
#Sta/Elev= 30
       0   72.58   62.27   72.53  120.53      72   260.3   71.62  260.85   71.81
  285.25   71.81  306.25   70.31  391.06   70.34  412.06   68.91  452.06   68.91
  473.06   70.41  566.41   70.43  587.41   71.93  611.82   71.93  613.12    71.5
  760.06    71.5  789.68   71.43  846.01      71 1048.08   71.47 1137.27   71.41
  1268.4   71.58 1358.38    71.5 1366.04      71 1373.51    69.5 1376.66      69
 1381.93    68.5 1399.68    68.5 1415.51    69.5 1430.31      70  1433.2   70.38
#Mann= 0 , 0 , 0
Levee=-1,285.33,71.8001,-1,587.45,71.93429,	340,	339
Bank Sta=391.06,473.06
XS Rating Curve= 0 ,0
Exp/Cntr=0.3,0.1

Type RM Length L Ch R = 1 ,7848.612,69.71,104.17,138.64
XS GIS Cut Line= 4
    1078856.8697    1572329.4841    1078785.7915    1572590.9508
    1078698.8347    1572878.1138    1078462.3223    1573660.4468
#Sta/Elev= 24
       0    72.5   78.19    72.5  138.34      72   269.6   71.56  271.41   71.56
  272.06   71.78  296.47   71.78  317.48   70.28  435.19   70.27  456.24    68.8
  496.27    68.8  517.26   70.27  526.77   70.27  547.78   71.77  572.19   71.77
  573.73   71.25  655.46   71.39   765.3      71 1195.07      71 1301.31   71.39
 1342.69    71.5  1378.2    71.5 1383.16      71  1388.3   70.16
#Mann= 0 , 0 , 0
Levee=-1,296.55,71.77283,-1,547.83,71.7709,	340,	339
Bank Sta=435.19,517.26
XS Rating Curve= 0 ,0
Exp/Cntr=0.3,0.1

Type RM Length L Ch R = 1 ,7744.441,136.14,96.57,56.98
XS GIS Cut Line= 6
     1078809.668    1572315.7257    1078755.1603    1572583.9023
    1078732.1978    1572678.9464    1078622.8718     1572729.903
    1078603.9276    1572741.1766    1078396.2822    1573647.3234
#Sta/Elev= 25
       0    72.5   83.96    72.5  143.29      72  272.73   71.52  273.01   71.52
  273.66   71.75  298.06   71.75  319.07   70.25  410.06    70.2  431.06   68.71
  471.06   68.71  491.13   70.14  492.06   70.14  581.73   70.12   602.7   71.61
  627.12   71.61  628.96      71 1011.28   70.92 1061.62   70.83 1120.55    70.9
 1178.58   70.85 1202.39      71  1318.7      71 1411.92    71.5 1443.73    71.5
#Mann= 0 , 0 , 0
Levee=-1,298.06,71.74581,-1,602.75,71.61491,	340,	339
Bank Sta=410.06,492.06
XS Rating Curve= 0 ,0
Exp/Cntr=0.3,0.1

Type RM Length L Ch R = 1 ,7647.875,123.11,84.42,45.74
XS GIS Cut Line= 4
     1078660.612     1572303.449    1078611.3139    1572552.2751
    1078568.3847    1572803.1983    1078364.2781    1573635.2584
#Sta/Elev= 24
       0   72.48  157.71    72.5  237.24      72  278.04   71.59  299.04   70.09
  308.61   70.09  329.93   68.61  369.98   68.62  390.79   70.09  508.24   70.09
  529.28   71.59  553.74   71.59   555.5      71  667.43      71  816.89   70.84
  924.02   70.85 1023.06   70.66 1052.44    70.7 1069.75   70.58  1085.2   70.59
  1159.5      71 1245.72      71 1296.12   71.28 1364.96    71.5
#Mann= 0 , 0 , 0
Levee=-1,278.06,71.58556,-1,529.34,71.58855,	340,	339
Bank Sta=308.61,390.79
XS Rating Curve= 0 ,0
Exp/Cntr=0.3,0.1

Type RM Length L Ch R = 1 ,7563.454,84.95,119.85,154.72
XS GIS Cut Line= 5
     1078506.095     1572265.349    1078465.0065    1572577.1945
     1078464.185    1572614.5997    1078546.1793     1572698.458
    1078316.2297    1573634.4117
#Sta/Elev= 25
       0      72   99.46      72  135.64   72.08  183.54   72.31  283.25      72
  286.83   71.91  314.49   69.93  387.24   69.97  388.18   69.97  408.24   68.54
  448.24   68.54  469.24   70.04  569.16   70.03  590.24   71.53  614.73   71.53
  616.32      71  680.66      71  878.59   70.71  970.01   70.71 1081.03    70.5
 1146.05    70.5 1249.41      71 1329.96      71 1405.85   71.16 1433.03   71.14
#Mann= 0 , 0 , 0
Levee=-1,293.57,71.42873,-1,590.23,71.52978,	340,	339
Bank Sta=387.24,469.24
XS Rating Curve= 0 ,0
Exp/Cntr=0.3,0.1

Type RM Length L Ch R = 1 ,7443.609,70.34,105.57,140.83
XS GIS Cut Line= 4
     1078465.455    1572258.3639    1078431.9017    1572573.9409
    1078412.4907    1572827.8406    1078269.2396    1573625.5217
#Sta/Elev= 23
       0      72  149.71      72  175.66   72.12   213.1      72  287.93      72
  317.36    69.9  434.41    69.9  455.37   68.43  494.12   68.42   495.7   68.42
  516.72    69.9  526.57    69.9  547.57    71.4  571.97    71.4  573.18      71
  746.15   70.57  824.51    70.5  1134.9    70.5 1164.56   70.83  1209.7      71
 1375.52      71 1378.08   70.81 1382.44   70.89
#Mann= 0 , 0 , 0
Levee=-1,296.43,71.39285,-1,547.59,71.40041,	340,	339
Bank Sta=434.41,516.72
XS Rating Curve= 0 ,0
Exp/Cntr=0.3,0.1

Type RM Length L Ch R = 1 ,7338.036,148.73,108.24,67.75
XS GIS Cut Line= 6
    1078440.6899    1572253.2839    1078410.0467     1572572.214
    1078402.5898    1572626.6647     1078303.739    1572699.4352
    1078288.2896    1572714.9299    1078224.1545    1573621.0767
#Sta/Elev= 20
       0      72  290.56      72  320.33   69.87  416.11   69.82  437.11   68.32
  477.11   68.32   497.2   69.76  498.11   69.76   581.1   69.74  602.14   71.24
  626.59   71.23  627.94   70.78  704.78    70.5 1215.23    70.5  1228.5   70.65
 1241.25   70.65 1295.63      71 1422.31      71 1425.83    70.5  1428.4   70.01
#Mann= 0 , 0 , 0
Levee=-1,299.31,71.37502,-1,602.22,71.23528,	340,	339
Bank Sta=416.11,498.11
XS Rating Curve= 0 ,0
Exp/Cntr=0.3,0.1

Type RM Length L Ch R = 1 ,7229.794,125.27,88.63,51.99
XS GIS Cut Line= 4
    1078259.0796    1572239.3139    1078248.9277    1572576.7524
    1078259.1448    1572775.2182    1078191.1344    1573617.9017
#Sta/Elev= 24
       0   71.59   29.72   71.63   101.6    71.5   154.3    71.5  240.12      72
   295.2      72  327.46    69.7  338.32    69.7  359.36   68.22   399.3   68.22
  420.26    69.7   536.9   69.71  557.97    71.2  582.45    71.2  583.94   70.71
   634.6    70.5 1196.78    70.5 1270.95      71 1357.37      71 1362.04    70.5
 1365.39      70 1372.89    68.5 1375.74      68 1381.74      68
#Mann= 0 , 0 , 0
Levee=-1,306.5,71.19247,-1,558.01,71.2039,	340,	339
Bank Sta=338.32,420.26
XS Rating Curve= 0 ,0
Exp/Cntr=0.3,0.1

Type RM Length L Ch R = 1 ,7141.164,78.58,113.31,148.04
XS GIS Cut Line= 6
    1078140.9693    1572227.8839    1078125.4875    1572526.2204
    1078118.7443    1572619.6797    1078212.2914    1572687.2832
    1078230.5045    1572701.5948    1078163.1944    1573616.6317
#Sta/Elev= 29
       0   71.18   43.91   71.07  140.93    71.5  219.06    71.5  285.94   71.99
  310.04      72  344.53   69.56  425.86   69.58  426.73   69.58  446.86   68.14
  486.86   68.14  507.86   69.64  605.87   69.66  626.97   71.16  651.49   71.16
  653.15   70.61  679.69    70.5 1281.23    70.5  1317.2    70.6 1325.42   70.69
 1340.26    70.5 1348.49    70.5 1355.67   70.63 1365.51   70.61 1412.31      71
 1426.23      71 1433.13      70 1442.11    68.5 1448.53    68.5
#Mann= 0 , 0 , 0
Levee=-1,323.4,71.05342,-1,626.99,71.16149,	340,	339
Bank Sta=425.86,507.86
XS Rating Curve= 0 ,0
Exp/Cntr=0.3,0.1

Type RM Length L Ch R = 1 ,7027.856,73.22,109.5,145.78
XS GIS Cut Line= 5
    1078089.5342    1572224.0739    1078072.2662    1572530.7353
    1078091.3989    1572692.3778    1078104.8158    1572829.0109
    1078096.5192    1573614.0916
#Sta/Elev= 30
       0      71   54.24      71  166.58    71.5  245.34    71.5  317.79   71.99
   352.5   69.51  469.92   69.51  490.89   68.03   530.9   68.03  551.91   69.51
  561.72   69.51  582.72   71.01  607.12   71.01  608.66    70.5  821.48   70.29
  838.62    70.5  903.76    70.5  911.13   70.42   973.2    70.5  988.04   70.16
 1023.09   70.42 1096.64   70.32 1177.09   70.38 1215.63    70.5 1341.61    70.5
 1366.45   70.69 1373.55   70.64 1377.63    70.5 1391.08    70.5 1392.33   70.34
#Mann= 0 , 0 , 0
Levee=-1,331.55,71.00288,-1,582.81,71.00985,	340,	339
Bank Sta=469.92,551.91
XS Rating Curve= 0 ,0
Exp/Cntr=0.3,0.1

Type RM Length L Ch R = 1 ,6918.354,130.83,93.53,56.23
XS GIS Cut Line= 6
    1078023.5364    1572218.3589    1078045.1515    1572579.2561
    1078058.2498    1572629.2047    1077972.8051    1572714.3585
    1077960.4596    1572730.8049    1078039.1998    1573628.6967
#Sta/Elev= 30
       0   70.88   79.45      71  181.95    71.5   263.3    71.5   326.9   71.94
  361.54   69.47  451.75   69.43  472.77   67.93   512.8   67.93  533.81   69.37
     626   69.34  647.09   70.84  671.59   70.84  673.27   70.29  673.92   70.28
  726.65   70.11  914.95      70  918.16   70.04  933.12   70.61  964.93   70.28
 1039.66      70 1071.76      70 1089.87   70.14 1190.63    70.1 1275.72    70.5
  1381.5    70.5  1401.9    69.8 1409.14   69.65 1422.37    69.6 1455.72   69.99
#Mann= 0 , 0 , 0
Levee=-1,340.59,70.9677,-1,647.12,70.84079,	340,	339
Bank Sta=451.75,533.81
XS Rating Curve= 0 ,0
Exp/Cntr=0.3,0.1

Type RM Length L Ch R = 1 ,6824.823,131.59,94.46,57.33
XS GIS Cut Line= 6
    1077850.8161    1572232.1172    1077906.1448    1572554.4187
    1077914.0826    1572610.7491     1077924.109    1572692.1077
    1077943.7248     1572852.662     1077993.903    1573633.3534
#Sta/Elev= 27
       0   70.25  159.44      71  235.22    71.5  341.95    71.5  372.44   69.32
   383.9   69.32  384.65   69.32  405.23   67.84  444.99   67.84  465.88   69.32
  582.12   69.31  603.17   70.81  627.63    70.8  629.35   70.24  629.69   70.23
  706.34   70.01  876.63      70  897.14    70.5 1031.73      70 1141.79      70
 1215.01   70.31 1242.65    70.5 1353.36    70.5  1360.6   70.41 1372.04      70
 1398.14      70 1409.93   70.15
#Mann= 0 , 0 , 0
Levee=-1,351.45,70.82193,-1,603.18,70.8055,	340,	339
Bank Sta=383.9,465.88
XS Rating Curve= 0 ,0
Exp/Cntr=0.3,0.1

Type RM Length L Ch R = 1 ,6730.362,79.99,110.99,142
XS GIS Cut Line= 6
    1077700.1091    1572245.6639    1077774.2871    1572583.9064
    1077790.7026    1572674.0781    1077886.8148    1572731.9604
    1077901.6162    1572740.9649    1077953.2629      1573641.82
#Sta/Elev= 28
       0      70  140.82      71  183.49    71.5  261.92    71.5  316.27   71.05
  369.58   70.71  391.74   69.18  467.69    69.2  468.57    69.2  488.81   67.76
  529.02   67.75  550.13   69.25  640.79   69.27  662.05   70.76  686.75   70.76
  688.56   70.16  744.64      70  963.13      70  981.52   70.21  1001.4   70.21
 1057.27      70 1230.67      70 1285.03   70.38 1319.17    70.5 1434.49    70.5
 1441.04   70.41  1451.4    70.5 1469.79    70.5
#Mann= 0 , 0 , 0
Levee=-1,370.74,70.6739,-1,662.07,70.76231,	340,	339
Bank Sta=467.69,550.13
XS Rating Curve= 0 ,0
Exp/Cntr=0.3,0.1

Type RM Length L Ch R = 1 ,6619.369,75.69,110.63,145.57
XS GIS Cut Line= 4
     1077636.609    1572260.0573    1077740.8731    1572639.9945
    1077809.3023    1572885.2722    1077905.0028    1573661.2934
#Sta/Elev= 22
       0      70   86.31   70.51   135.2      71  143.89      71  180.33    71.3
  277.49   71.26  358.27   70.63     373   70.63  393.98   69.13  512.11   69.13
  533.12   67.65  573.12   67.65  594.11   69.13   603.2   69.13   624.2   70.63
   648.6   70.63  650.08   70.14  715.19      70 1183.83      70 1277.34   70.41
 1326.95    70.5 1430.53    70.5
#Mann= 0 , 0 , 0
Levee=-1,373.04,70.6272,-1,624.23,70.62787,	340,	339
Bank Sta=512.11,594.11
XS Rating Curve= 0 ,0
Exp/Cntr=0.3,0.1

Type RM Length L Ch R = 1 ,6508.738,137.26,95.23,53.18
XS GIS Cut Line= 6
    1077584.9622     1572271.064    1077696.0224    1572605.9842
    1077725.5092    1572696.9381    1077659.7331    1572797.3003
    1077647.6157    1572818.8584    1077849.1227    1573670.6068
#Sta/Elev= 19
       0   69.95   99.18   70.52  170.27   71.02  196.52   71.12  306.69   71.01
  377.18   70.59  398.18   69.09  486.46   69.05  507.46   67.55  547.46   67.55
  567.62   68.99  568.46   68.99   662.1   68.95  683.28   70.45     851      70
 1302.36      70 1363.21   70.13 1431.57    70.5 1468.45    70.5
#Mann= 0 , 0 , 0
Levee=-1,377.26,70.58814,-1,683.35,70.45036,	340,	339
Bank Sta=486.46,568.46
XS Rating Curve= 0 ,0
Exp/Cntr=0.3,0.1

Type RM Length L Ch R = 1 ,6413.504,134.85,98.46,62.09
XS GIS Cut Line= 5
    1077443.5686    1572310.0107    1077551.8597    1572656.1842
     1077611.188    1572780.7703    1077628.1423    1572851.8785
     1077822.876    1573686.6935
#Sta/Elev= 24
       0   69.78  136.03    70.5  197.96      71  379.14      71  408.15   68.93
  418.07   68.93  439.24   67.46  479.53   67.46  500.71   68.94  618.79   68.92
  640.57   70.45  773.68   70.21  827.62      70 1214.78      70 1230.26   69.87
 1239.88      70 1322.84      70 1353.98   70.14 1368.61    70.5 1373.65    70.5
 1382.39   70.25  1396.7   70.33 1401.82    70.5 1431.03    70.5
#Mann= 0 , 0 , 0
Levee=-1,387.18,70.42523,-1,640.1,70.4221,	340,	339
Bank Sta=418.07,500.71
XS Rating Curve= 0 ,0
Exp/Cntr=0.3,0.1

Type RM Length L Ch R = 1 ,6315.049,74.08,109.52,144.96
XS GIS Cut Line= 6
    1077313.1817    1572370.9708    1077423.2416    1572712.0683
     1077468.122    1572801.0784    1077576.7283    1572827.4692
    1077593.4289    1572833.2518    1077788.1626    1573701.9335
#Sta/Elev= 30
       0   70.21   42.21    70.5  123.98    70.5  178.76   70.67  269.18    70.5
  335.58   70.99  373.42   70.97   403.8   68.78  487.87   68.81  508.87   67.37
  548.87   67.37  569.87   68.87  663.35   68.88  687.15   70.55  798.33   70.37
  917.92      70 1230.29      70 1276.63    69.5 1318.59    69.5 1329.37      70
  1392.6      70 1399.85    70.2 1405.43      70 1416.39      70 1428.89   70.31
 1432.59    70.5 1448.72    70.5 1457.27      70 1469.02   68.77 1477.78   68.39
#Mann= 0 , 0 , 0
Levee=-1,382.82,70.27781,-1,684.77,70.3833,	340,	339
Bank Sta=487.87,569.87
XS Rating Curve= 0 ,0
Exp/Cntr=0.3,0.1
